HEC-RAS study Howards Creek.prj: Howards Creek Limited Detail Study

--- Howards Creek.g01 (geometry) --- (continued)

Type RM Length L Ch R =3,32395,,,
BEGIN DESCRIPTION:
Howards Creek Mill Rd TOR HC
Structure ID: LDS_HC_06
Approximate Survey Structure
END DESCRIPTION:
Bridge Culvert--1,0,-1,-1,0
Deck Dist Width WeirC Skew NumUp NumDn MinLoCord MaxHiCord MaxSubmerge Is_Ogee
16.5,25,3,,43,43,,,,0,1,1,,,
  4606.8  4626.7  4670.4  4678.7  4764.0  4771.5  4842.9  4866.9  4873.7  4930.0
  4955.0  4955.0  5045.0  5045.0  5081.1  5092.6  5100.7  5111.8  5150.3  5153.3
  5159.7  5160.5  5197.3  5203.8  5210.7  5215.5  5223.1  5238.0  5239.1  5247.5
  5249.4  5269.4  5287.0  5300.8  5303.1  5306.2  5320.0  5335.3  5335.5  5347.7
  5360.0  5363.9  5378.9
  867.93  866.47  862.67  862.19  854.61  853.50  847.57  846.04  845.35  842.80
  842.80  842.80  842.80  842.80  842.80  842.98  842.87  843.07  843.71  843.77
  843.72  843.74  845.03  844.66  845.13  845.20  845.81  846.93  846.98  848.41
  848.94  854.79  857.83  858.81  858.89  859.31  861.60  863.07  863.08  864.82
  867.11  867.58  869.63
  808.20  808.20  808.20  808.20  808.20  808.20  808.20  808.20  808.20  808.20
  808.20  840.30  840.30  808.20  808.20  808.20  808.20  808.20  808.20  808.20
  808.20  808.20  808.20  808.20  808.20  808.20  808.20  808.20  808.20  808.20
  808.20  808.20  808.20  808.20  808.20  808.20  808.20  808.20  808.20  808.20
  808.20  808.20  808.20
  4606.8  4626.7  4670.4  4678.7  4764.0  4771.5  4842.9  4866.9  4873.7  4930.0
  4955.0  4955.0  5045.0  5045.0  5081.1  5092.6  5100.7  5111.8  5150.3  5153.3
  5159.7  5160.5  5197.3  5203.8  5210.7  5215.5  5223.1  5238.0  5239.1  5247.5
  5249.4  5269.4  5287.0  5300.8  5303.1  5306.2  5320.0  5335.3  5335.5  5347.7
  5360.0  5363.9  5378.9
  867.93  866.47  862.67  862.19  854.61  853.50  847.57  846.04  845.35  842.80
  842.80  842.80  842.80  842.80  842.80  842.98  842.87  843.07  843.71  843.77
  843.72  843.74  845.03  844.66  845.13  845.20  845.81  846.93  846.98  848.41
  848.94  854.79  857.83  858.81  858.89  859.31  861.60  863.07  863.08  864.82
  867.11  867.58  869.63
  808.20  808.20  808.20  808.20  808.20  808.20  808.20  808.20  808.20  808.20
  808.20  840.30  840.30  808.20  808.20  808.20  808.20  808.20  808.20  808.20
  808.20  808.20  808.20  808.20  808.20  808.20  808.20  808.20  808.20  808.20
  808.20  808.20  808.20  808.20  808.20  808.20  808.20  808.20  808.20  808.20
  808.20  808.20  808.20
Pier Skew, UpSta & Num, DnSta & Num=,4977.5,2,4977.5,2,0,0,0,0,0
       1       1
  830.91  840.30
       1       1
  830.66  840.30
Pier Skew, UpSta & Num, DnSta & Num=,5022.5,2,5022.5,2,0,0,0,0,0
       1       1
  830.83  840.30
       1       1
  830.58  840.30
BR Coef=1,1,0,1.25,0,,,0.8,0,2,0,
WSPro=,,,, 1 ,,,, 0 ,,,, 0 ,,,,-1 ,-1 ,-1 , 0 , 0 , 0 , 0 , 0
BC Design=,,0,,0,,,,,,

Type RM Length L Ch R = 1,32350,325,325,325
BEGIN DESCRIPTION:
Howards Creek Mill Rd d/s HC
END DESCRIPTION:
XS GIS Cut Line= 6
      1294825.46       645663.65      1294691.64       645597.63
      1294586.36       645551.23      1294518.55       645522.68
      1294484.65       645479.86      1294452.53       645362.09
#Sta/Elev= 30
  4632.1  869.23  4655.3  868.96  4663.2  867.94  4703.1  860.44  4707.6  860.42
  4738.5  853.81  4761.5  849.76  4776.7  846.12  4796.4  843.07  4820.9  841.91
  4830.6  840.61  4837.7  840.63  4855.0  842.44  4863.5  842.26  4877.5  841.36
  4895.9  838.28  4919.3  837.50  4932.9  836.25  4948.2  836.88  4955.3  835.93
  4968.4  837.40  4980.8  827.20  5019.3  827.20  5031.7  837.40  5043.3  835.76
  5078.2  842.70  5098.5  848.58  5108.7  849.50  5131.6  854.10  5146.7  855.33
#Mann=3,-1,0
  4632.1    0.15       0  4968.4   0.045       0  5031.7    0.15       0
#XS Ineff=2,0
    0.00 4922.50  843.14 5077.50    0.00  842.80
Bank Sta=4968.4,5031.7
XS Rating Curve= 0
Exp/Cntr=0.5,0.3

Type RM Length L Ch R = 1,32025,490,490,490
BEGIN DESCRIPTION:
Howards Creek 64.0
END DESCRIPTION:
XS GIS Cut Line= 3
      1294879.67       645670.23      1294806.02       645336.69
      1294518.34       645174.10
#Sta/Elev= 30
  4591.6  874.88  4619.8  870.26  4632.5  869.63  4659.5  866.10  4705.2  858.86
  4810.1  846.66  4822.5  845.98  4909.6  833.61  4922.4  833.93  4927.1  832.52
  4933.1  832.73  4953.7  830.26  4963.6  827.86  4964.6  826.64  4964.7  827.23
  4987.3  826.64  4988.8  823.64  5011.2  823.64  5012.7  826.64  5015.6  833.85
  5050.2  833.92  5099.0  838.89  5118.7  843.27  5126.9  843.59  5135.6  847.19
  5167.9  854.83  5184.1  857.23  5237.5  867.30  5248.1  867.16  5263.6  870.85
#Mann=3,-1,0
  4591.6    0.15       0  4987.3    0.05       0  5012.7    0.15       0
Bank Sta=4987.3,5012.7
XS Rating Curve= 0
Exp/Cntr=0.3,0.1

Type RM Length L Ch R = 1,31535,693,693,693
BEGIN DESCRIPTION:
Howards Creek 63.0
END DESCRIPTION:
XS GIS Cut Line= 3
      1295058.99       645573.05      1295186.00       645200.13
      1295207.62       645070.42
#Sta/Elev= 30
  4654.8  857.35  4680.0  854.61  4715.7  853.09  4732.0  851.64  4759.6  848.36
  4811.2  840.85  4848.1  833.09  4920.5  833.43  4939.9  833.08  4953.7  833.70
  4960.9  832.82  4966.4  831.44  4978.3  825.15  4980.0  824.75  4984.5  826.13
  4986.6  822.86  4988.1  819.86  5011.9  819.86  5013.4  822.86  5018.8  832.06
  5044.1  841.78  5055.4  843.37  5068.6  847.74  5086.5  852.11  5096.6  853.20
  5109.5  855.30  5132.0  857.49  5141.3  858.77  5156.3  859.87  5180.3  863.21
#Mann=3,-1,0
  4654.8    0.15       0  4986.6    0.05       0  5013.4    0.15       0
Bank Sta=4986.6,5013.4
XS Rating Curve= 0
Exp/Cntr=0.3,0.1

Type RM Length L Ch R = 1,30842,438,438,438
BEGIN DESCRIPTION:
Howards Creek 62.0
END DESCRIPTION:
XS GIS Cut Line= 2
      1295775.00       645825.00      1295894.00       645078.53
#Sta/Elev= 30
  4548.6  881.59  4635.6  867.39  4658.6  862.38  4682.2  855.30  4718.4  841.72
  4747.6  831.65  4764.5  829.48  4782.8  828.40  4805.5  829.43  4853.5  829.48
  4887.6  828.74  4902.3  829.68  4934.3  827.76  4946.3  828.81  4959.0  828.51
  4972.6  826.76  4984.1  818.66  4985.8  819.81  4986.6  818.66  4988.1  815.66
  5011.9  815.66  5013.4  818.66  5018.0  827.82  5066.3  827.99  5111.8  826.80
  5142.9  827.27  5170.6  831.48  5222.2  846.39  5267.6  858.72  5304.5  867.29
#Mann=3,-1,0
  4548.6    0.15       0  4986.6    0.05       0  5013.4    0.15       0
Bank Sta=4986.6,5013.4
XS Rating Curve= 0
Exp/Cntr=0.3,0.1

Type RM Length L Ch R = 1,30404,497,497,497
BEGIN DESCRIPTION:
Howards Creek 61.0
END DESCRIPTION:
XS GIS Cut Line= 3
      1296153.42       645805.45      1296269.62       645435.23
      1296326.37       645375.78
#Sta/Elev= 30
  4675.4  850.00  4747.6  841.48  4760.1  840.76  4774.4  839.29  4789.5  838.80
  4801.5  837.36  4830.1  836.41  4854.8  835.92  4860.4  835.19  4865.1  834.89
  4873.1  834.86  4886.0  832.84  4898.7  831.23  4910.8  828.33  4922.3  825.93
  4952.9  825.43  4960.0  820.81  4971.6  815.54  4977.5  816.33  4986.6  815.54
  4988.1  812.54  5011.9  812.54  5013.4  815.54  5016.3  819.21  5046.3  825.06
  5058.7  825.46  5065.5  827.53  5082.9  832.28  5105.3  839.98  5145.6  851.01
#Mann=3,-1,0
  4675.4    0.15       0  4986.6    0.05       0  5013.4    0.15       0
Bank Sta=4986.6,5013.4
XS Rating Curve= 0
Exp/Cntr=0.3,0.1

Type RM Length L Ch R = 1,29907,373,373,373
BEGIN DESCRIPTION:
Howards Creek 60.0
END DESCRIPTION:
XS GIS Cut Line= 2
      1296504.72       645808.15      1296796.57       645648.72
#Sta/Elev= 24
  4797.7  844.71  4882.6  834.15  4894.3  833.26  4947.6  823.98  4954.6  823.28
  4968.0  823.13  4970.7  823.52  4985.7  818.24  4986.6  815.17  4988.1  812.17
  5011.9  812.17  5013.4  815.17  5016.5  816.48  5031.1  822.70  5031.7  822.95
  5032.0  823.10  5032.3  823.26  5046.9  830.73  5051.5  833.65  5072.9  848.44
  5082.4  853.22  5105.9  862.09  5117.5  866.04  5130.3  869.71
#Mann=3,-1,0
  4797.7    0.15       0  4986.6    0.05       0  5013.4    0.15       0
Bank Sta=4986.6,5013.4
XS Rating Curve= 0
Exp/Cntr=0.3,0.1

Type RM Length L Ch R = 1,29534,214,214,214
BEGIN DESCRIPTION:
Howards Creek 59.5
END DESCRIPTION:
XS GIS Cut Line= 3
      1296541.30       646018.90      1296720.53       646086.35
      1296809.17       646088.28
#Sta/Elev= 30
  4844.4  838.33  4862.0  836.20  4871.5  834.51  4878.3  833.91  4886.1  832.88
  4900.4  830.30  4907.4  828.79  4921.4  826.30  4934.0  824.42  4958.3  821.38
  4963.6  821.43  4968.8  821.97  4976.5  822.26  4985.0  822.14  4986.6  814.13
  4988.1  811.13  5011.9  811.13  5013.4  814.13  5025.3  815.06  5026.7  815.36
  5035.9  817.82  5062.6  824.61  5071.2  827.44  5083.9  832.00  5085.6  832.45
  5099.9  836.90  5113.1  840.90  5119.2  842.05  5123.5  843.69  5124.5  843.97
#Mann=3,-1,0
  4844.4    0.15       0  4986.6    0.05       0  5013.4    0.15       0
Bank Sta=4986.6,5013.4
XS Rating Curve= 0
Exp/Cntr=0.3,0.1

Type RM Length L Ch R = 1,29320,320,320,320
BEGIN DESCRIPTION:
Howards Creek 59.0
END DESCRIPTION:
XS GIS Cut Line= 2
      1296489.27       646425.52      1296855.43       646144.16
#Sta/Elev= 30
  4765.9  875.20  4792.1  868.92  4861.3  849.15  4888.0  839.73  4912.6  830.67
  4932.2  822.19  4935.2  821.61  4942.5  821.04  4953.3  819.66  4964.8  818.99
  4967.1  816.93  4972.3  813.06  4981.3  813.95  4986.6  813.06  4988.1  810.06
  5011.9  810.06  5013.4  813.06  5024.4  816.05  5038.9  817.95  5053.5  821.23
  5083.9  826.62  5117.1  830.94  5135.3  833.85  5153.3  837.77  5165.9  839.02
  5177.2  840.92  5189.4  841.53  5200.7  842.76  5223.8  846.49  5227.6  847.45
#Mann=3,-1,0
  4765.9    0.15       0  4986.6    0.05       0  5013.4    0.15       0
Bank Sta=4986.6,5013.4
XS Rating Curve= 0
Exp/Cntr=0.3,0.1

Type RM Length L Ch R = 1,29000,301,301,301
BEGIN DESCRIPTION:
Howards Creek 58.0
END DESCRIPTION:
XS GIS Cut Line= 3
      1296925.00       646525.00      1296979.14       646337.28
      1297025.00       646225.00
#Sta/Elev= 30
  4804.6  850.50  4822.7  846.57  4835.2  844.37  4845.6  842.15  4852.2  841.06
  4855.8  840.19  4868.1  838.09  4881.5  834.99  4896.0  832.01  4911.3  828.29
  4925.4  825.10  4934.9  821.76  4939.0  819.83  4943.4  819.23  4953.5  817.43
  4958.8  812.43  4968.6  811.04  4971.2  810.86  4986.6  810.99  4988.1  807.99
  5011.9  807.99  5013.4  810.99  5020.5  812.17  5030.7  816.13  5038.9  817.74
  5059.4  823.86  5061.8  824.35  5066.2  825.89  5105.6  838.18  5121.3  842.17
#Mann=3,-1,0
  4804.6    0.15       0  4986.6    0.05       0  5013.4    0.12       0
Bank Sta=4986.6,5013.4
XS Rating Curve= 0
Exp/Cntr=0.3,0.1

Type RM Length L Ch R = 1,28699,127,127,127
BEGIN DESCRIPTION:
Howard Creek 57.5
END DESCRIPTION:
XS GIS Cut Line= 2
      1297226.36       646590.05      1297312.78       646236.28
#Sta/Elev= 29
  4818.7  851.22  4846.0  846.17  4855.4  844.18  4867.9  841.18  4887.2  835.11
  4888.5  834.65  4890.1  834.15  4893.5  832.95  4901.6  830.23  4924.6  821.91
  4928.7  820.26  4936.6  816.34  4937.8  813.14  4945.0  812.59  4950.2  812.62
  4961.8  810.53  4986.6  809.04  4988.1  806.04  5011.9  806.04  5013.4  809.04
  5037.3  821.72  5074.5  828.66  5076.9  829.00  5085.1  831.13  5090.5  832.34
  5111.3  836.40  5121.5  838.93  5148.7  843.86  5182.9  848.34
#Mann=3,-1,0
  4818.7    0.15       0  4986.6    0.05       0  5013.4     0.1       0
Bank Sta=4986.6,5013.4
XS Rating Curve= 0
Exp/Cntr=0.5,0.3

Type RM Length L Ch R = 1,28572,54,54,54
BEGIN DESCRIPTION:
SR 1193 u/s HC
END DESCRIPTION:
XS GIS Cut Line= 6
      1297304.38       646629.51      1297370.02       646564.89
      1297383.36       646500.27      1297392.59       646423.35
      1297420.28       646283.86      1297399.77       646201.81
#Sta/Elev= 30
  4795.1  851.61  4829.4  844.96  4841.4  842.06  4844.2  840.63  4864.6  835.11
  4870.0  832.83  4884.3  829.11  4896.3  826.81  4908.4  825.12  4925.3  823.87
  4940.2  821.43  4953.9  816.78  4976.0  810.90  4981.5  805.20  5018.5  805.20
  5024.0  810.90  5030.7  814.59  5056.7  820.71  5064.5  823.60  5095.5  828.58
  5106.7  830.00  5118.3  830.93  5134.8  833.42  5146.1  834.66  5156.5  835.22
  5167.2  836.55  5177.7  837.12  5215.3  842.84  5240.7  845.14  5257.4  847.25
#Mann=3,-1,0
  4795.1    0.15       0  4976.0    0.05       0  5024.0     0.1       0
#XS Ineff=2,0
    0.00 4946.00  818.02 5054.00    0.00  825.05
Bank Sta=4976,5024
XS Rating Curve= 0
Exp/Cntr=0.5,0.3

Type RM Length L Ch R =3,28549,,,
BEGIN DESCRIPTION:
SR 1193 TOR HC
Structure ID: LDS_HC_05
Approximate Survey Structure
END DESCRIPTION:
Bridge Culvert--1,0,-1,-1,0
Deck Dist Width WeirC Skew NumUp NumDn MinLoCord MaxHiCord MaxSubmerge Is_Ogee
14,18,3,,45,45,,,,0,1,1,,,
  4671.5  4710.7  4723.5  4727.5  4737.1  4757.3  4791.6  4803.1  4808.7  4821.4
  4823.3  4825.2  4830.8  4836.8  4839.9  4849.0  4858.3  4861.4  4880.6  4885.4
  4889.1  4929.9  4942.7  4960.0  4960.0  5040.0  5040.0  5045.9  5047.0  5062.6
  5071.4  5075.0  5090.1  5093.6  5096.3  5103.7  5113.9  5124.8  5207.9  5209.6
  5226.5  5228.9  5230.9  5240.0  5258.8
  865.29  862.76  861.32  860.72  858.98  855.70  848.87  844.41  842.94  838.98
  838.46  837.67  835.74  833.53  832.65  829.48  828.97  828.68  827.38  827.27
  826.94  824.94  824.55  824.50  824.50  824.50  824.50  824.85  825.04  825.06
  826.07  826.60  827.50  827.45  827.81  828.13  829.00  829.67  836.66  836.90
  838.63  838.81  839.03  839.76  841.57
  785.20  785.20  785.20  785.20  785.20  785.20  785.20  785.20  785.20  785.20
  785.20  785.20  785.20  785.20  785.20  785.20  785.20  785.20  785.20  785.20
  785.20  785.20  785.20  785.20  822.00  822.00  785.20  785.20  785.20  785.20
  785.20  785.20  785.20  785.20  785.20  785.20  785.20  785.20  785.20  785.20
  785.20  785.20  785.20  785.20  785.20
  4671.5  4710.7  4723.5  4727.5  4737.1  4757.3  4791.6  4803.1  4808.7  4821.4
  4823.3  4825.2  4830.8  4836.8  4839.9  4849.0  4858.3  4861.4  4880.6  4885.4
  4889.1  4929.9  4942.7  4960.0  4960.0  5040.0  5040.0  5045.9  5047.0  5062.6
  5071.4  5075.0  5090.1  5093.6  5096.3  5103.7  5113.9  5124.8  5207.9  5209.6
  5226.5  5228.9  5230.9  5240.0  5258.8
  865.29  862.76  861.32  860.72  858.98  855.70  848.87  844.41  842.94  838.98
  838.46  837.67  835.74  833.53  832.65  829.48  828.97  828.68  827.38  827.27
  826.94  824.94  824.55  824.50  824.50  824.50  824.50  824.85  825.04  825.06
  826.07  826.60  827.50  827.45  827.81  828.13  829.00  829.67  836.66  836.90
  838.63  838.81  839.03  839.76  841.57
  785.20  785.20  785.20  785.20  785.20  785.20  785.20  785.20  785.20  785.20
  785.20  785.20  785.20  785.20  785.20  785.20  785.20  785.20  785.20  785.20
  785.20  785.20  785.20  785.20  822.00  822.00  785.20  785.20  785.20  785.20
  785.20  785.20  785.20  785.20  785.20  785.20  785.20  785.20  785.20  785.20
  785.20  785.20  785.20  785.20  785.20
Pier Skew, UpSta & Num, DnSta & Num=,5000,2,5000,2,0,0,0,0,0
       1       1
  805.20  822.00
       1       1
  804.95  822.00
BR Coef=1,1,0,1.25,0,,,0.8,0,2,0,
WSPro=,,,, 1 ,,,, 0 ,,,, 0 ,,,,-1 ,-1 ,-1 , 0 , 0 , 0 , 0 , 0
BC Design=,,0,,0,,,,,,

Type RM Length L Ch R = 1,28518,124,124,124
BEGIN DESCRIPTION:
SR 1193 d/s HC
END DESCRIPTION:
XS GIS Cut Line= 5
      1297536.18       646759.77      1297416.18       646600.79
      1297436.69       646482.84      1297464.38       646395.66
      1297535.15       646231.55
#Sta/Elev= 30
  4672.1  839.07  4687.8  835.28  4701.8  828.97  4718.9  823.27  4749.6  818.73
  4782.5  817.79  4819.4  819.55  4826.8  821.94  4838.9  820.23  4843.4  826.44
  4850.8  828.85  4887.7  828.16  4941.5  823.33  4948.6  820.22  4951.2  816.93
  4965.2  811.99  4966.7  812.84  4976.0  810.65  4981.5  804.95  5018.5  804.95
  5024.0  810.65  5025.8  816.56  5047.8  822.75  5071.1  824.15  5088.8  827.11
  5102.3  827.50  5177.6  837.57  5216.5  840.51  5228.5  842.98  5261.2  845.65
#Mann=3,-1,0
  4672.1    0.15       0  4976.0    0.05       0  5024.0     0.1       0
#XS Ineff=2,0
    0.00 4938.00  824.69 5062.00    0.00  825.06
Bank Sta=4976,5024
XS Rating Curve= 0
Exp/Cntr=0.5,0.3

Type RM Length L Ch R = 1,28394,394,394,394
BEGIN DESCRIPTION:
Howards Creek 57.0
END DESCRIPTION:
XS GIS Cut Line= 3
      1297577.54       646779.63      1297537.00       646644.51
      1297591.05       646312.13
#Sta/Elev= 30
  4718.3  848.97  4741.4  846.16  4752.3  843.40  4765.5  842.29  4772.7  840.98
  4781.4  836.40  4801.8  827.25  4853.5  818.32  4903.1  815.46  4920.8  815.17
  4930.8  813.90  4949.5  810.47  4954.9  808.98  4958.5  809.36  4963.8  806.32
  4969.4  805.62  4973.5  805.36  4977.9  805.63  4986.6  806.84  4988.1  803.84
  5011.9  803.84  5013.4  806.84  5018.7  814.57  5025.6  816.64  5037.7  820.99
  5075.1  829.69  5133.1  837.28  5150.3  838.83  5161.8  840.47  5196.1  841.14
#Mann=3,-1,0
  4718.3    0.15       0  4986.6    0.05       0  5013.4     0.1       0
Bank Sta=4986.6,5013.4
XS Rating Curve= 0
Exp/Cntr=0.3,0.1

Type RM Length L Ch R = 1,28000,525,525,525
BEGIN DESCRIPTION:
Howards Creek 56.0
END DESCRIPTION:
XS GIS Cut Line= 3
      1297961.26       646411.03      1297887.30       646346.47
      1297769.40       646259.71
#Sta/Elev= 25
  4901.8  827.46  4908.5  824.06  4911.7  822.49  4923.7  816.08  4928.3  813.32
  4935.7  810.24  4938.5  809.16  4948.1  807.33  4948.5  807.10  4949.7  801.43
  4966.2  802.52  4978.9  802.40  4983.4  802.21  4986.6  801.43  4988.1  798.43
  5011.9  798.43  5013.4  801.43  5071.7  822.77  5079.1  824.44  5095.5  828.82
  5103.8  829.98  5124.4  833.34  5134.3  835.34  5142.8  836.83  5146.4  837.09
#Mann=3,-1,0
  4901.8    0.15       0  4986.6    0.05       0  5013.4     0.1       0
Bank Sta=4986.6,5013.4
XS Rating Curve= 0
Exp/Cntr=0.3,0.1

Type RM Length L Ch R = 1,27475,475,475,475
BEGIN DESCRIPTION:
Howards Creek 55.0
END DESCRIPTION:
XS GIS Cut Line= 3
      1298336.88       646097.57      1298299.05       646019.20
      1298199.06       645851.66
#Sta/Elev= 20
  4924.4  829.32  4985.6  796.84  4987.1  793.84  5012.9  793.84  5014.4  796.84
  5016.8  799.08  5064.4  805.62  5077.7  806.65  5087.3  807.10  5106.8  809.21
  5120.3  809.94  5136.9  811.68  5148.4  813.58  5154.9  814.91  5160.7  815.92
  5169.9  817.18  5188.8  820.10  5202.8  822.72  5206.0  823.23  5206.6  823.34
#Mann=3,-1,0
  4924.4    0.15       0  4985.6    0.05       0  5014.4    0.15       0
Bank Sta=4985.6,5014.4
XS Rating Curve= 0
Exp/Cntr=0.3,0.1

Type RM Length L Ch R = 1,27000,544,544,544
BEGIN DESCRIPTION:
Howards Creek 54.0
END DESCRIPTION:
XS GIS Cut Line= 3
      1298753.03       646021.90      1298731.22       645836.63
      1298685.48       645662.50
#Sta/Elev= 30
  4813.4  822.22  4856.5  817.00  4871.9  814.29  4887.6  811.97  4904.9  808.89
  4915.6  807.35  4932.7  805.76  4968.3  803.69  4974.0  803.57  4978.5  802.74
  4985.6  794.20  4987.1  791.20  5012.9  791.20  5014.4  794.20  5020.0  794.56
  5022.6  795.43  5026.4  797.77  5031.3  801.91  5034.1  802.42  5042.8  802.48
  5054.3  802.86  5065.9  804.06  5069.9  805.63  5090.5  815.92  5102.2  821.09
  5108.9  823.20  5120.5  825.01  5128.3  825.38  5173.9  830.84  5180.0  831.73
#Mann=3,-1,0
  4813.4     0.1       0  4985.6    0.05       0  5014.4    0.15       0
Bank Sta=4985.6,5014.4
XS Rating Curve= 0
Exp/Cntr=0.3,0.1

Type RM Length L Ch R = 1,26456,577,577,577
BEGIN DESCRIPTION:
Howards Creek 53.0
END DESCRIPTION:
XS GIS Cut Line= 3
      1299312.41       645698.98      1299209.72       645647.63
      1298828.70       645466.58
#Sta/Elev= 30
  4918.3  836.28  4921.8  833.74  4946.8  818.70  4965.7  804.33  4976.7  797.46
  4982.6  795.10  4985.3  794.61  4985.6  793.23  4987.1  790.23  5012.9  790.23
  5014.4  793.23  5018.1  794.59  5028.1  797.23  5038.5  799.39  5046.2  799.13
  5060.6  800.83  5074.2  800.74  5097.7  803.19  5137.9  805.94  5144.7  805.97
  5157.2  806.80  5178.7  807.47  5264.7  808.62  5322.0  811.22  5362.5  814.97
  5380.5  815.60  5396.0  817.14  5403.0  817.49  5433.6  820.22  5454.9  823.00
#Mann=3,-1,0
  4918.3    0.15       0  4985.6    0.05       0  5014.4    0.15       0
Bank Sta=4985.6,5014.4
XS Rating Curve= 0
Exp/Cntr=0.3,0.1

Type RM Length L Ch R = 1,25879,379,379,379
BEGIN DESCRIPTION:
Howards Creek 52.0
END DESCRIPTION:
XS GIS Cut Line= 2
      1299528.59       645199.05      1298998.94       644820.73
#Sta/Elev= 30
  4856.9  830.07  4877.0  826.09  4920.3  815.03  4953.2  801.01  4959.2  800.45
  4976.8  793.19  4985.6  790.83  4987.1  787.83  5012.9  787.83  5014.4  790.83
  5017.7  793.13  5030.0  799.35  5143.4  798.69  5152.4  797.85  5209.8  796.81
  5229.1  797.60  5248.4  797.73  5261.2  797.03  5300.1  797.96  5306.9  797.22
  5319.7  798.21  5325.6  797.92  5366.8  799.23  5377.7  800.51  5398.1  800.09
  5422.2  803.08  5444.1  810.25  5457.0  812.67  5476.0  819.10  5507.8  828.36
#Mann=3,-1,0
  4856.9    0.15       0  4985.6    0.05       0  5014.4    0.15       0
Bank Sta=4985.6,5014.4
XS Rating Curve= 0
Exp/Cntr=0.3,0.1

Type RM Length L Ch R = 1,25500,716,716,716
BEGIN DESCRIPTION:
Howards Creek 51.0
END DESCRIPTION:
XS GIS Cut Line= 3
      1299652.90       645184.19      1299668.35       644841.31
      1299612.37       644495.10
#Sta/Elev= 30
  4656.8  837.59  4711.5  827.00  4740.9  820.33  4760.5  814.74  4780.1  806.87
  4798.2  802.46  4813.8  799.82  4847.7  797.53  4902.5  798.54  4947.0  798.03
  4985.6  789.29  4987.1  786.29  5012.9  786.29  5014.4  789.29  5018.9  795.12
  5023.3  794.98  5030.7  798.27  5092.7  796.27  5138.2  796.57  5152.7  797.69
  5165.1  797.73  5168.7  798.37  5186.5  807.82  5212.8  817.26  5242.9  826.52
  5289.8  835.74  5316.8  838.10  5330.6  838.59  5342.0  840.06  5350.7  840.07
#Mann=3,-1,0
  4656.8    0.15       0  4985.6    0.05       0  5014.4    0.15       0
Bank Sta=4985.6,5014.4
XS Rating Curve= 0
Exp/Cntr=0.3,0.1

Type RM Length L Ch R = 1,24784,434,434,434
BEGIN DESCRIPTION:
Howards Creek 50.0
END DESCRIPTION:
XS GIS Cut Line= 3
      1300514.93       644976.11      1300198.76       644392.42
      1299904.21       644095.16
#Sta/Elev= 30
  4280.5  823.01  4327.5  817.05  4347.1  816.77  4362.6  813.94  4390.4  812.11
  4420.7  808.48  4496.5  796.84  4520.5  794.54  4569.7  792.39  4591.8  793.49
  4658.6  792.61  4734.7  793.95  4831.3  793.30  4927.9  794.76  4985.6  787.04
  4987.1  784.04  5012.9  784.04  5014.4  787.04  5015.1  792.04  5027.8  795.61
  5092.3  793.82  5166.9  794.50  5190.3  793.11  5208.8  794.23  5224.6  799.89
  5231.4  804.34  5262.0  819.31  5281.5  825.61  5299.9  828.82  5362.8  836.56
#Mann=3,-1,0
  4280.5    0.15       0  4985.6    0.05       0  5014.4    0.15       0
Bank Sta=4985.6,5014.4
XS Rating Curve= 0
Exp/Cntr=0.3,0.1

Type RM Length L Ch R = 1,24350,495,495,495
BEGIN DESCRIPTION:
Howards Creek 49.0
END DESCRIPTION:
XS GIS Cut Line= 3
      1300906.77       644483.21      1300506.83       644131.92
      1300279.83       643904.92
#Sta/Elev= 30
  4416.5  822.01  4452.5  813.24  4470.0  808.14  4506.7  794.95  4529.2  791.15
  4548.8  790.62  4592.8  791.12  4598.0  792.15  4614.5  791.31  4644.6  791.02
  4682.6  791.96  4710.3  791.45  4769.7  792.40  4833.8  791.88  4911.5  793.65
  4980.0  787.95  4985.6  786.01  4987.1  783.01  5012.9  783.01  5014.4  786.01
  5033.2  791.15  5044.3  792.35  5079.2  794.06  5108.4  793.01  5149.6  793.47
  5154.8  794.04  5192.1  808.24  5224.8  818.41  5244.6  822.19  5269.8  825.82
#Mann=3,-1,0
  4416.5    0.15       0  4985.6    0.05       0  5014.4    0.15       0
Bank Sta=4985.6,5014.4
XS Rating Curve= 0
Exp/Cntr=0.3,0.1

Type RM Length L Ch R = 1,23855,174,174,174
BEGIN DESCRIPTION:
Howards Creek 48.0
END DESCRIPTION:
XS GIS Cut Line= 4
      1300966.22       644307.57      1300967.52       644190.81
      1300831.10       643872.50      1300647.35       643540.11
#Sta/Elev= 30
  4643.1  817.62  4660.9  816.02  4710.8  809.85  4747.6  806.79  4761.0  806.56
  4802.3  799.12  4808.5  798.98  4825.1  794.85  4849.9  791.21  4940.3  791.26
  4954.6  790.01  4985.6  783.33  4987.1  780.33  5012.9  780.33  5014.4  783.33
  5014.6  784.09  5028.9  784.41  5068.3  791.80  5140.6  790.95  5244.7  790.94
  5262.1  790.13  5270.4  790.83  5321.2  790.76  5336.2  792.16  5344.6  792.21
  5362.1  793.61  5378.1  796.45  5394.9  801.70  5432.1  811.94  5486.0  819.54
#Mann=3,-1,0
  4643.1    0.15       0  4985.6    0.05       0  5014.4     0.1       0
Bank Sta=4985.6,5014.4
XS Rating Curve= 0
Exp/Cntr=0.3,0.1

Type RM Length L Ch R = 1,23681,213,213,213
BEGIN DESCRIPTION:
Howards Creek 47.5
END DESCRIPTION:
XS GIS Cut Line= 3
      1300979.73       644283.24      1301009.45       644021.12
      1301090.52       643772.51
#Sta/Elev= 30
  4649.6  816.31  4669.0  813.72  4675.4  812.37  4683.8  811.96  4692.2  810.89
  4728.2  808.14  4736.3  808.04  4749.6  806.84  4776.6  805.34  4863.8  796.93
  4891.7  793.00  4914.5  791.01  4925.9  790.75  4933.4  791.38  4941.6  791.25
  4953.5  791.60  4967.4  790.92  4981.5  788.40  4989.3  783.29  4992.0  780.11
  5009.1  780.11  5010.8  783.11  5016.3  788.91  5045.0  796.85  5079.0  807.85
  5111.8  815.40  5128.7  818.34  5148.8  823.39  5159.8  825.45  5174.8  828.88
#Mann=3,-1,0
  4649.6    0.15       0  4989.3    0.06       0  5010.8    0.15       0
Bank Sta=4989.3,5010.8
XS Rating Curve= 0
Exp/Cntr=0.3,0.1

Type RM Length L Ch R = 1,23468,459,459,459
BEGIN DESCRIPTION:
Howards Creek 47.0
END DESCRIPTION:
XS GIS Cut Line= 3
      1300975.00       644325.00      1301214.83       644048.14
      1301301.30       643731.98
#Sta/Elev= 30
  4553.4  820.97  4580.0  817.16  4603.2  811.40  4624.6  807.13  4659.9  797.73
  4678.1  794.09  4704.9  790.12  4746.4  790.05  4832.7  792.30  4843.9  791.69
  4856.3  789.21  4876.3  790.15  4882.6  787.92  4888.5  786.85  4901.5  786.39
  4930.3  787.62  4951.6  789.69  4963.8  788.48  4975.0  783.74  4979.6  783.69
  4985.9  782.14  4987.9  778.89  5004.6  778.88  5006.3  781.89  5067.3  790.75
  5120.2  793.89  5150.2  804.62  5159.8  808.80  5188.3  815.43  5247.4  827.25
#Mann=3,-1,0
  4553.4     0.2       0  4985.9    0.06       0  5006.3     0.2       0
#XS Ineff=2,0
    0.00 4833.70  801.88               0
Bank Sta=4985.9,5006.3
XS Rating Curve= 0
Exp/Cntr=0.3,0.1

Type RM Length L Ch R = 1,23009,494,494,494
BEGIN DESCRIPTION:
Howards Creek 46.0
END DESCRIPTION:
XS GIS Cut Line= 3
      1301112.14       644508.89      1301349.94       644365.66
      1301531.00       644352.15
#Sta/Elev= 30
  4671.1  819.90  4685.9  817.06  4699.0  815.04  4707.8  813.98  4734.0  808.36
  4762.3  803.46  4813.6  797.97  4845.3  795.96  4849.6  795.82  4856.3  796.72
  4862.9  796.80  4875.4  797.57  4887.1  797.31  4904.8  794.10  4919.3  793.18
  4951.6  790.01  4962.6  788.00  4971.9  782.84  4985.7  780.98  4988.8  777.98
  5012.2  777.98  5014.5  780.98  5015.8  788.82  5019.4  789.89  5030.6  790.93
  5052.3  791.25  5095.8  802.55  5111.5  807.03  5120.4  808.68  5130.2  811.27
#Mann=3,-1,0
  4671.1    0.15       0  4985.7    0.45       0  5014.5    0.15       0
Bank Sta=4985.7,5014.5
XS Rating Curve= 0
Exp/Cntr=0.3,0.1

Type RM Length L Ch R = 1,22515,515,515,515
BEGIN DESCRIPTION:
Howards Creek 45.0
END DESCRIPTION:
XS GIS Cut Line= 3
      1301379.67       644995.30      1301395.88       644735.88
      1301468.84       644630.49
#Sta/Elev= 30
  4816.6  820.87  4834.9  818.25  4863.3  813.26  4871.9  811.96  4892.5  807.39
  4896.1  806.30  4914.2  802.05  4918.1  800.62  4938.2  794.38  4947.2  791.87
  4960.3  789.87  4975.5  788.37  4978.3  788.49  4985.6  779.32  4987.1  776.32
  5012.9  776.32  5014.4  779.32  5025.0  784.91  5029.7  785.74  5065.4  790.24
  5076.5  790.82  5088.8  790.48  5106.1  790.56  5119.3  791.61  5150.3  795.64
  5158.7  796.43  5178.4  798.75  5191.4  800.83  5200.4  801.52  5204.7  802.45
#Mann=3,-1,0
  4816.6    0.12       0  4985.6    0.45       0  5014.4    0.15       0
Bank Sta=4985.6,5014.4
XS Rating Curve= 0
Exp/Cntr=0.3,0.1

Type RM Length L Ch R = 1,22000,228,228,228
BEGIN DESCRIPTION:
Howards Creek 44.0
END DESCRIPTION:
XS GIS Cut Line= 3
      1301809.33       644968.28      1301873.19       644773.78
      1301925.00       644675.00
#Sta/Elev= 26
  4795.3  815.16  4800.3  814.18  4813.2  812.42  4858.5  804.58  4867.0  802.83
  4895.3  796.84  4904.0  795.26  4927.5  788.89  4931.7  788.17  4940.3  787.08
  4949.0  787.11  4952.6  787.03  4955.2  787.13  4968.9  788.58  4971.8  788.46
  4980.3  784.95  4985.6  777.06  4987.1  774.06  5012.9  774.06  5014.4  777.06
  5034.4  788.81  5036.7  790.34  5038.9  790.62  5073.9  801.35  5100.7  810.76
  5111.5  813.19
#Mann=3,-1,0
  4795.3    0.12       0  4985.6    0.05       0  5014.4    0.15       0
Bank Sta=4985.6,5014.4
XS Rating Curve= 0
Exp/Cntr=0.3,0.1

Type RM Length L Ch R = 1,21772,151,151,151
BEGIN DESCRIPTION:
Howards Creek 43.5
END DESCRIPTION:
XS GIS Cut Line= 2
      1302012.01       645146.63      1302117.40       644676.43
#Sta/Elev= 30
  4728.9  820.42  4741.5  818.33  4804.2  810.51  4819.0  807.98  4832.2  806.64
  4844.0  804.56  4847.7  803.22  4879.9  799.20  4911.1  793.57  4916.3  792.03
  4924.4  790.42  4967.4  786.59  4979.9  785.02  4984.9  785.22  4985.6  776.96
  4987.1  773.96  5012.9  773.96  5014.4  776.96  5025.7  782.25  5041.6  784.21
  5055.0  787.76  5069.7  788.01  5082.4  790.13  5093.6  793.92  5114.5  800.01
  5147.9  807.80  5163.5  811.93  5177.7  814.50  5205.8  820.73  5210.7  821.64
#Mann=3,-1,0
  4728.9    0.12       0  4985.6    0.06       0  5014.4    0.15       0
Bank Sta=4985.6,5014.4
XS Rating Curve= 0
Exp/Cntr=0.3,0.1

Type RM Length L Ch R = 1,21621,121,121,121
BEGIN DESCRIPTION:
Howards Creek 43.2
END DESCRIPTION:
XS GIS Cut Line= 4
      1302119.78       645178.12      1302218.05       644992.51
      1302221.69       644839.65      1302156.17       644694.07
#Sta/Elev= 30
  4679.0  809.30  4711.3  802.10  4727.8  798.92  4734.2  798.09  4776.7  789.72
  4796.7  787.37  4813.4  786.49  4854.3  786.80  4931.0  785.62  4938.9  786.95
  4941.6  787.72  4947.9  787.62  4949.0  787.92  4962.6  788.63  4975.9  784.73
  4982.2  779.51  4983.4  779.22  4985.6  776.96  4987.1  773.96  5012.9  773.96
  5014.4  776.96  5018.9  778.21  5081.8  792.71  5101.6  793.51  5119.5  796.07
  5132.8  798.50  5151.5  803.01  5159.3  805.38  5174.4  808.40  5201.5  814.82
#Mann=3,-1,0
  4679.0    0.12       0  4985.6    0.05       0  5014.4    0.15       0
Bank Sta=4985.6,5014.4
XS Rating Curve= 0
Exp/Cntr=0.3,0.1

Type RM Length L Ch R = 1,21500,363,363,363
BEGIN DESCRIPTION:
Howards Creek 43.0
END DESCRIPTION:
XS GIS Cut Line= 3
      1302575.00       645675.00      1302333.78       644845.60
      1302175.00       644675.00
#Sta/Elev= 30
  4136.2  826.09  4230.1  818.47  4237.8  816.88  4283.6  813.14  4345.0  804.58
  4420.9  791.67  4431.7  790.60  4464.3  788.91  4518.6  788.95  4547.3  790.07
  4611.8  789.72  4649.8  788.10  4662.3  788.75  4791.7  788.80  4824.2  786.72
  4868.8  787.40  4924.9  786.47  4961.3  787.66  4978.2  783.50  4983.6  778.15
  4985.6  776.95  4987.1  773.95  5012.9  773.95  5014.4  776.95  5017.4  776.95
  5030.0  781.87  5043.7  784.45  5059.3  783.87  5138.3  792.10  5233.1  816.19
#Mann=3,-1,0
  4136.2    0.15       0  4985.6    0.06       0  5014.4    0.15       0
Bank Sta=4985.6,5014.4
XS Rating Curve= 0
Exp/Cntr=0.3,0.1

Type RM Length L Ch R = 1,21137,763,763,763
BEGIN DESCRIPTION:
Howards Creek 42.0
END DESCRIPTION:
XS GIS Cut Line= 3
      1302778.52       645578.46      1302720.29       644770.50
      1302367.26       644370.16
#Sta/Elev= 30
  4060.9  820.41  4182.7  804.17  4205.1  798.32  4267.1  787.63  4306.5  783.80
  4321.7  785.78  4347.8  784.69  4419.8  785.99  4508.5  784.57  4579.8  785.75
  4605.4  783.86  4628.9  786.25  4657.1  784.62  4712.1  785.28  4726.0  783.39
  4744.2  786.07  4955.8  787.13  4985.6  776.91  4987.1  773.91  5012.9  773.91
  5014.4  776.91  5018.1  780.91  5047.1  785.43  5156.9  783.68  5224.9  784.83
  5263.1  787.49  5307.8  793.45  5331.1  799.43  5374.5  806.08  5404.7  812.73
#Mann=3,-1,0
  4060.9    0.15       0  4985.6    0.05       0  5014.4    0.15       0
Bank Sta=4985.6,5014.4
XS Rating Curve= 0
Exp/Cntr=0.3,0.1

Type RM Length L Ch R = 1,20374,207,207,207
BEGIN DESCRIPTION:
Howards Creek 41.0
END DESCRIPTION:
XS GIS Cut Line= 3
      1303425.00       644725.00      1303325.32       644307.57
      1302974.02       643988.69
#Sta/Elev= 30
  4675.8  804.27  4698.1  804.47  4724.2  800.60  4778.2  786.06  4815.5  782.67
  4833.6  778.29  4858.6  781.99  4935.6  781.76  4951.6  783.74  4961.5  784.25
  4985.6  776.59  4987.1  773.59  5012.9  773.59  5014.4  776.59  5028.2  783.73
  5058.5  784.33  5071.7  785.36  5100.3  783.69  5117.9  783.89  5132.1  782.99
  5140.7  783.70  5221.1  782.05  5287.5  782.47  5318.2  781.41  5329.4  782.40
  5451.0  782.71  5487.4  782.06  5541.4  798.13  5563.8  801.70  5579.4  804.95
#Mann=3,-1,0
  4675.8    0.12       0  4985.6    0.05       0  5014.4    0.15       0
#XS Ineff=2,0
       0                 5280.00    0.00  789.80
Bank Sta=4985.6,5014.4
XS Rating Curve= 0
Exp/Cntr=0.5,0.3

Type RM Length L Ch R = 1,20167,70,70,70
BEGIN DESCRIPTION:
Alf Hoover Road u/s HC
END DESCRIPTION:
XS GIS Cut Line= 6
      1303541.51       644680.48      1303533.81       644443.50
      1303550.20       644380.28      1303543.18       644287.20
      1303498.27       644077.87      1303498.27       643929.24
#Sta/Elev= 30
  4665.3  808.83  4816.4  796.89  4828.6  795.56  4849.7  791.49  4868.0  788.95
  4883.3  788.22  4899.0  788.94  4918.9  787.04  4929.2  784.80  4975.5  784.10
  4984.8  773.50  5015.3  773.50  5024.5  784.10  5033.3  780.97  5048.3  783.25
  5059.1  782.99  5087.9  784.28  5099.5  783.60  5161.9  783.94  5192.6  785.94
  5219.0  782.58  5265.1  780.36  5288.6  782.73  5294.5  783.87  5332.1  787.25
  5342.2  789.33  5353.2  792.55  5359.9  795.58  5375.7  799.31  5424.2  804.15
#Mann=3,-1,0
  4665.3    0.12       0  4975.5    0.05       0  5024.5    0.15       0
#XS Ineff=2,0
    0.00 4918.80  790.49 5081.30    0.00  790.28
Bank Sta=4975.5,5024.5
XS Rating Curve= 0
Exp/Cntr=0.5,0.3

Type RM Length L Ch R =3,20130,,,
BEGIN DESCRIPTION:
Alf Hoover Road TOR HC
Structure ID: LDS_HC_04
Approximate Survey Structure
END DESCRIPTION:
Bridge Culvert--1,0,-1,-1,0
Deck Dist Width WeirC Skew NumUp NumDn MinLoCord MaxHiCord MaxSubmerge Is_Ogee
27,20,3,,38,38,,,,0,1,1,,,
  4665.6  4729.0  4734.4  4743.6  4747.7  4754.6  4760.3  4764.9  4768.0  4776.7
  4787.6  4788.1  4823.2  4875.0  4890.4  4928.9  4936.2  4945.8  4945.8  5054.3
  5054.3  5074.1  5104.7  5113.3  5130.6  5220.0  5227.3  5230.7  5235.7  5238.1
  5310.8  5320.8  5331.3  5334.8  5339.4  5342.2  5350.9  5361.3
  808.09  803.21  801.39  801.79  801.42  799.63  798.89  797.91  797.77  797.67
  795.48  795.44  793.78  791.65  791.40  790.16  790.21  790.20  790.20  790.20
  790.20  790.29  790.24  790.46  790.46  793.72  794.32  794.61  794.78  794.78
  799.78  800.21  800.93  801.28  801.45  801.82  802.17  802.99
  753.50  753.50  753.50  753.50  753.50  753.50  753.50  753.50  753.50  753.50
  753.50  753.50  753.50  753.50  753.50  753.50  753.50  753.50  788.50  788.50
  753.50  753.50  753.50  753.50  753.50  753.50  753.50  753.50  753.50  753.50
  753.50  753.50  753.50  753.50  753.50  753.50  753.50  753.50
  4665.6  4729.0  4734.4  4743.6  4747.7  4754.6  4760.3  4764.9  4768.0  4776.7
  4787.6  4788.1  4823.2  4875.0  4890.4  4928.9  4936.2  4945.8  4945.8  5054.3
  5054.3  5074.1  5104.7  5113.3  5130.6  5220.0  5227.3  5230.7  5235.7  5238.1
  5310.8  5320.8  5331.3  5334.8  5339.4  5342.2  5350.9  5361.3
  808.09  803.21  801.39  801.79  801.42  799.63  798.89  797.91  797.77  797.67
  795.48  795.44  793.78  791.65  791.40  790.16  790.21  790.20  790.20  790.20
  790.20  790.29  790.24  790.46  790.46  793.72  794.32  794.61  794.78  794.78
  799.78  800.21  800.93  801.28  801.45  801.82  802.17  802.99
  753.50  753.50  753.50  753.50  753.50  753.50  753.50  753.50  753.50  753.50
  753.50  753.50  753.50  753.50  753.50  753.50  753.50  753.50  788.50  788.50
  753.50  753.50  753.50  753.50  753.50  753.50  753.50  753.50  753.50  753.50
  753.50  753.50  753.50  753.50  753.50  753.50  753.50  753.50
Pier Skew, UpSta & Num, DnSta & Num=,4972.9,2,4972.9,2,0,0,0,0,0
       1       1
  784.26  788.50
       1       1
  784.37  788.50
Pier Skew, UpSta & Num, DnSta & Num=,5027.1,2,5027.1,2,0,0,0,0,0
       1       1
  783.18  788.50
       1       1
  783.15  788.50
BR Coef=1,1,0,1.25,0,,,0.8,0,2,0,
WSPro=,,,, 1 ,,,, 0 ,,,, 0 ,,,,-1 ,-1 ,-1 , 0 , 0 , 0 , 0 , 0
BC Design=,,0,,0,,,,,,

Type RM Length L Ch R = 1,20097,173,173,173
BEGIN DESCRIPTION:
Alf Hoover Road d/s HC
END DESCRIPTION:
XS GIS Cut Line= 5
      1303660.41       644653.46      1303641.49       644442.68
      1303614.60       644328.18      1303624.73       644245.64
      1303622.58       643980.59
#Sta/Elev= 30
  4669.8  807.02  4719.5  804.56  4745.5  802.01  4801.7  793.20  4822.9  791.66
  4854.3  786.36  4900.9  785.20  4920.8  783.81  4940.7  784.80  4950.8  783.61
  4957.9  784.56  4964.6  783.91  4973.8  784.42  4975.5  783.85  4984.8  773.25
  5015.3  773.25  5024.5  783.85  5045.1  778.27  5050.2  778.73  5063.9  784.57
  5095.2  784.01  5109.0  784.59  5137.4  782.99  5207.4  781.51  5237.2  782.99
  5282.6  794.34  5298.8  801.06  5311.1  803.51  5336.6  810.70  5347.3  813.00
#Mann=3,-1,0
  4669.8    0.15       0  4975.5    0.05       0  5024.5    0.15       0
#XS Ineff=2,0
    0.00 4922.80  790.36 5077.30    0.00  790.28
Bank Sta=4975.5,5024.5
XS Rating Curve= 0
Exp/Cntr=0.5,0.3

Type RM Length L Ch R = 1,19924,291,291,291
BEGIN DESCRIPTION:
Howards Creek 40.0
END DESCRIPTION:
XS GIS Cut Line= 3
      1303702.77       644711.95      1303783.49       644337.01
      1303747.04       643988.10
#Sta/Elev= 30
  4546.6  808.36  4605.6  808.14  4626.3  807.21  4641.9  805.52  4661.9  801.84
  4686.1  796.53  4716.1  791.78  4734.5  790.26  4795.2  787.41  4816.8  785.40
  4824.9  785.31  4838.7  783.62  4935.8  782.12  4946.1  782.17  4961.1  783.60
  4970.7  783.60  4985.6  775.31  4987.1  772.31  5012.9  772.31  5014.4  775.31
  5066.4  783.48  5086.1  782.23  5116.8  782.46  5136.3  780.08  5146.0  780.18
  5168.6  781.71  5192.5  785.86  5196.7  785.90  5246.2  801.30  5280.9  810.36
#Mann=3,-1,0
  4546.6    0.15       0  4985.6    0.05       0  5014.4    0.15       0
Bank Sta=4985.6,5014.4
XS Rating Curve= 0
Exp/Cntr=0.3,0.1

Type RM Length L Ch R = 1,19633,603,603,603
BEGIN DESCRIPTION:
Howards Creek 39.0
END DESCRIPTION:
XS GIS Cut Line= 3
      1303940.28       644799.33      1304010.00       644666.22
      1304054.37       643848.58
#Sta/Elev= 30
  4324.9  809.36  4345.1  807.30  4358.8  806.82  4597.4  801.15  4631.6  797.44
  4682.3  793.94  4720.0  788.87  4730.4  788.89  4741.7  789.98  4798.3  788.21
  4826.2  785.29  4838.4  782.53  4854.0  781.48  4884.8  782.07  4925.1  781.79
  4967.8  774.86  4985.6  773.77  4987.1  770.77  5012.9  770.77  5014.4  773.77
  5019.8  782.71  5021.2  783.79  5094.6  781.80  5106.0  782.34  5127.3  785.65
  5180.8  799.62  5195.9  802.18  5212.1  806.11  5242.7  810.91  5294.0  821.31
#Mann=3,-1,0
  4324.9    0.15       0  4985.6    0.05       0  5014.4    0.15       0
Bank Sta=4985.6,5014.4
XS Rating Curve= 0
Exp/Cntr=0.3,0.1

Type RM Length L Ch R = 1,19030,339,339,339
BEGIN DESCRIPTION:
Howards Creek 38.0
END DESCRIPTION:
XS GIS Cut Line= 2
      1304618.48       644336.63      1304453.69       643538.00
#Sta/Elev= 30
  4411.6  793.92  4488.1  790.69  4504.9  790.32  4542.0  786.49  4583.4  783.24
  4634.0  781.10  4663.4  780.99  4689.7  779.48  4698.5  779.88  4729.3  780.06
  4762.2  779.83  4773.6  779.46  4784.2  778.49  4838.5  778.50  4854.6  778.12
  4943.2  779.83  4950.7  779.28  4985.6  772.04  4987.1  769.04  5012.9  769.04
  5014.4  772.04  5023.2  774.98  5072.9  780.11  5085.5  779.41  5096.0  779.84
  5133.7  788.59  5150.8  790.67  5180.6  795.18  5205.8  798.07  5227.1  802.26
#Mann=3,-1,0
  4411.6    0.15       0  4985.6    0.05       0  5014.4    0.15       0
Bank Sta=4985.6,5014.4
XS Rating Curve= 0
Exp/Cntr=0.3,0.1

Type RM Length L Ch R = 1,18691,400,400,400
BEGIN DESCRIPTION:
Howards Creek 37.0
END DESCRIPTION:
XS GIS Cut Line= 3
      1304967.09       643911.96      1304878.35       643645.75
      1304517.07       643322.50
#Sta/Elev= 30
  4541.6  797.52  4596.1  796.39  4688.1  793.35  4778.0  789.34  4814.7  788.49
  4848.0  786.57  4860.0  783.64  4870.7  783.04  4884.6  781.19  4893.1  779.53
  4927.7  780.61  4960.3  773.35  4985.6  771.38  4987.1  768.38  5012.9  768.38
  5014.4  771.38  5049.9  781.84  5066.5  780.81  5099.3  781.52  5158.1  779.14
  5181.1  780.17  5191.4  779.76  5207.8  780.47  5214.2  782.87  5218.2  782.35
  5235.3  785.81  5249.5  789.36  5289.8  792.80  5295.1  793.79  5307.0  797.43
#Mann=3,-1,0
  4541.6    0.15       0  4985.6    0.05       0  5014.4    0.15       0
Bank Sta=4985.6,5014.4
XS Rating Curve= 0
Exp/Cntr=0.3,0.1

Type RM Length L Ch R = 1,18291,861,861,861
BEGIN DESCRIPTION:
Howards Creek 36.0
END DESCRIPTION:
XS GIS Cut Line= 4
      1305493.17       643918.30      1305268.71       643527.32
      1305000.46       643225.54      1304547.79       643236.72
#Sta/Elev= 30
  4241.7  815.51  4299.9  813.82  4365.1  809.83  4417.4  804.43  4452.1  798.92
  4487.4  795.12  4545.0  790.44  4557.2  788.55  4610.2  784.49  4671.1  784.07
  4696.6  781.97  4704.1  780.62  4749.0  778.41  4856.3  778.64  4867.5  778.08
  4901.0  779.12  4941.2  778.16  4958.1  780.44  4963.2  777.84  4973.1  777.20
  4985.6  771.25  4987.1  768.25  5012.9  768.25  5014.4  771.25  5061.1  780.88
  5125.6  778.04  5332.7  779.03  5490.8  778.50  5508.0  780.61  5549.1  795.93
#Mann=3,-1,0
  4241.7    0.15       0  4985.6    0.05       0  5014.4    0.15       0
Bank Sta=4985.6,5014.4
XS Rating Curve= 0
Exp/Cntr=0.3,0.1

Type RM Length L Ch R = 1,17430,430,430,430
BEGIN DESCRIPTION:
Howards Creek 35.0
END DESCRIPTION:
XS GIS Cut Line= 4
      1305727.69       644051.41      1305833.14       643664.24
      1305894.62       643544.09      1305841.78       642891.50
#Sta/Elev= 30
  4414.5  812.57  4659.8  799.78  4670.0  798.19  4697.1  795.81  4721.5  791.43
  4735.9  790.43  4784.9  778.37  4823.3  777.19  4858.3  777.96  4894.4  777.27
  4953.5  777.81  4975.3  776.15  4986.4  773.38  4989.5  769.65  4992.1  766.65
  5010.7  766.65  5013.3  769.65  5021.5  772.62  5030.1  776.82  5048.5  778.29
  5078.9  778.14  5095.8  777.27  5164.0  783.76  5220.5  787.46  5347.0  801.63
  5381.7  803.65  5426.1  807.84  5486.9  810.43  5533.6  809.90  5605.4  812.22
#Mann=3,-1,0
  4414.5    0.15       0  4989.5    0.06       0  5013.3    0.15       0
Bank Sta=4989.5,5013.3
XS Rating Curve= 0
Exp/Cntr=0.3,0.1

Type RM Length L Ch R = 1,17000,500,500,500
BEGIN DESCRIPTION:
Howards Creek 34.0
END DESCRIPTION:
XS GIS Cut Line= 3
      1305975.00       644425.00      1306320.31       643513.29
      1306298.14       642111.88
#Sta/Elev= 30
  4025.1  821.32  4142.3  802.73  4166.2  799.90  4179.2  796.42  4192.3  794.41
  4217.7  787.02  4249.7  774.43  4299.9  773.40  4672.9  775.25  4929.2  776.90
  4979.1  778.86  4984.7  769.18  4986.2  766.18  5013.8  766.18  5015.3  769.18
  5022.9  770.73  5090.7  774.47  5107.3  773.64  5330.0  773.76  5385.4  772.64
  5420.7  774.14  5610.2  772.03  5640.6  773.31  5713.6  771.93  6019.2  776.91
  6111.5  781.00  6177.8  782.25  6303.4  788.93  6320.9  790.68  6401.6  793.37
#Mann=3,-1,0
  4025.1    0.15       0  4984.7    0.05       0  5015.3    0.15       0
Bank Sta=4984.7,5015.3
XS Rating Curve= 0
Exp/Cntr=0.3,0.1

Type RM Length L Ch R = 1,16500,500,500,500
BEGIN DESCRIPTION:
Howards Creek 33.0
END DESCRIPTION:
XS GIS Cut Line= 3
      1306525.00       644775.00      1306819.28       643544.31
      1307217.19       642200.62
#Sta/Elev= 30
  3734.6  823.64  3802.7  818.20  3855.8  810.65  3932.8  795.14  4008.5  774.41
  4079.6  771.62  4298.0  771.91  4517.4  773.69  4632.0  773.36  4961.1  776.33
  4984.7  767.70  4986.2  764.70  5013.8  764.70  5015.3  767.70  5035.6  769.10
  5060.6  776.06  5165.6  773.30  5241.9  773.01  5265.8  771.46  5334.0  773.37
  5459.4  771.48  5535.5  773.32  5755.1  774.35  5961.3  777.37  5971.8  777.28
  5982.9  775.36  5986.7  778.56  6004.6  780.23  6117.4  783.20  6401.4  801.32
#Mann=3,-1,0
  3734.6    0.08       0  4984.7    0.05       0  5015.3    0.12       0
Bank Sta=4984.7,5015.3
XS Rating Curve= 0
Exp/Cntr=0.3,0.1

Type RM Length L Ch R = 1,16000,500,500,500
BEGIN DESCRIPTION:
Howards Creek 32.0
END DESCRIPTION:
XS GIS Cut Line= 3
      1306805.20       644779.68      1307316.75       643580.44
      1307469.46       642457.32
#Sta/Elev= 30
  3696.2  805.42  3827.2  795.36  3870.0  784.40  3900.4  778.21  3964.1  771.80
  4551.1  773.81  4564.7  773.49  4578.8  770.93  4589.8  773.22  4909.0  773.59
  4984.7  767.40  4986.2  764.40  5013.8  764.40  5015.3  767.40  5039.7  773.57
  5044.5  776.24  5048.5  776.31  5181.7  772.86  5222.1  773.70  5253.0  771.77
  5349.9  772.84  5418.3  771.30  5498.6  772.61  5550.1  771.84  5760.8  775.39
  5771.4  774.61  5774.4  776.29  5844.7  777.07  5924.5  783.79  6133.4  793.05
#Mann=3,-1,0
  3696.2    0.08       0  4984.7    0.05       0  5015.3    0.12       0
Bank Sta=4984.7,5015.3
XS Rating Curve= 0
Exp/Cntr=0.3,0.1

Type RM Length L Ch R = 1,15500,500,500,500
BEGIN DESCRIPTION:
Howards Creek 31.0
END DESCRIPTION:
XS GIS Cut Line= 3
      1308036.36       644378.59      1307815.70       643576.52
      1307517.12       642528.82
#Sta/Elev= 30
  4168.1  797.44  4324.3  793.10  4370.1  788.19  4436.8  771.87  4488.4  771.58
  4527.7  773.28  4648.7  771.28  4687.7  773.02  4760.4  771.42  4925.7  772.13
  4967.9  773.54  4979.9  766.69  4981.4  763.69  5018.6  763.69  5020.1  766.69
  5026.9  768.48  5035.9  767.70  5060.1  775.21  5123.3  771.92  5220.8  772.99
  5234.0  771.04  5243.7  773.39  5288.2  771.75  5412.9  771.55  5646.1  775.84
  5728.5  774.55  5754.0  777.92  5821.6  778.21  5953.9  782.87  6089.4  789.74
#Mann=3,-1,0
  4168.1    0.15       0  4979.9    0.05       0  5020.1    0.12       0
Bank Sta=4979.9,5020.1
XS Rating Curve= 0
Exp/Cntr=0.3,0.1

Type RM Length L Ch R = 1,15000,665,665,665
BEGIN DESCRIPTION:
Howards Creek 30.0
END DESCRIPTION:
XS GIS Cut Line= 4
      1308291.92       644163.60      1308315.29       643573.69
      1308097.20       643141.35      1308052.58       642796.55
#Sta/Elev= 30
  4409.6  804.88  4534.3  800.29  4586.6  796.28  4616.0  793.35  4656.5  785.30
  4683.6  782.44  4724.5  775.41  4743.1  772.91  4774.5  770.58  4786.0  771.25
  4836.0  770.35  4935.3  771.97  4962.9  773.34  4979.9  766.18  4981.4  763.18
  5018.6  763.18  5020.1  766.18  5037.0  773.56  5054.7  773.32  5079.0  771.86
  5130.5  772.53  5176.9  771.03  5202.5  772.48  5227.9  776.42  5261.8  778.67
  5301.0  783.76  5324.6  785.10  5463.1  780.01  5726.4  784.73  5831.9  787.81
#Mann=3,-1,0
  4409.6     0.1       0  4979.9    0.05       0  5020.1     0.1       0
Bank Sta=4979.9,5020.1
XS Rating Curve= 0
Exp/Cntr=0.3,0.1

Type RM Length L Ch R = 1,14335,286,286,286
BEGIN DESCRIPTION:
Howards Creek 29.0
END DESCRIPTION:
XS GIS Cut Line= 3
      1308855.77       644200.10      1309115.39       642897.96
      1309125.00       642675.00
#Sta/Elev= 30
  4361.3  799.33  4399.2  795.45  4441.3  789.63  4472.1  784.09  4514.2  780.13
  4547.7  775.69  4593.8  773.43  4667.9  772.37  4743.6  773.18  4786.6  771.12
  4833.2  771.17  4856.4  769.39  4901.0  770.90  4923.6  770.49  4966.8  772.78
  4979.9  765.96  4981.4  762.96  5018.6  762.96  5020.1  765.96  5045.6  773.22
  5138.7  772.00  5197.9  770.04  5299.5  769.16  5547.7  769.09  5741.9  771.64
  5762.6  775.41  5801.0  791.41  5830.4  802.09  5878.0  811.75  5912.2  817.20
#Mann=3,-1,0
  4361.3     0.1       0  4979.9    0.05       0  5020.1     0.1       0
Bank Sta=4979.9,5020.1
XS Rating Curve= 0
Exp/Cntr=0.3,0.1

Type RM Length L Ch R = 1,14049,292,292,292
BEGIN DESCRIPTION:
Howards Creek 28.0
END DESCRIPTION:
XS GIS Cut Line= 3
      1309143.46       644085.47      1309226.54       643714.21
      1309427.74       642995.32
#Sta/Elev= 30
  4470.6  786.98  4537.1  785.18  4614.4  781.14  4646.9  777.38  4658.7  774.38
  4670.9  772.66  4697.1  770.43  4736.9  770.03  4756.2  768.62  4833.8  770.78
  4866.7  770.62  4877.7  769.55  4921.0  770.85  4950.8  770.46  4979.1  772.46
  4979.9  765.88  4981.4  762.88  5018.6  762.88  5020.1  765.88  5031.6  770.93
  5057.2  773.13  5095.2  770.82  5377.8  770.39  5396.8  768.91  5430.6  769.27
  5449.4  771.13  5471.2  775.56  5522.6  783.14  5560.9  797.09  5597.6  805.31
#Mann=3,-1,0
  4470.6     0.1       0  4979.9    0.05       0  5020.1     0.1       0
#XS Ineff=2,0
    0.00 4701.40  780.08 5304.10    0.00  780.08
Bank Sta=4979.9,5020.1
XS Rating Curve= 0
Exp/Cntr=0.5,0.3

Type RM Length L Ch R = 1,13757,78,78,78
BEGIN DESCRIPTION:
Daniels Road u/s HC
END DESCRIPTION:
XS GIS Cut Line= 6
      1309120.10       644150.37      1309379.71       643833.64
      1309540.10       643600.39      1309578.07       643522.27
      1309595.20       643402.67      1309688.66       643187.19
#Sta/Elev= 30
  4265.2  790.70  4287.6  789.13  4317.5  788.60  4347.6  786.44  4392.1  785.66
  4468.7  779.84  4583.5  772.51  4674.8  770.52  4725.4  771.19  4784.1  770.20
  4842.7  771.11  4935.8  771.32  4941.4  772.22  4970.8  769.63  4977.8  770.55
  4983.8  762.80  5016.3  762.80  5022.3  770.55  5024.7  769.34  5033.3  770.79
  5063.3  770.41  5075.1  771.31  5113.0  772.07  5140.0  771.71  5228.9  778.32
  5241.2  778.77  5262.6  781.31  5295.8  787.01  5336.5  790.78  5400.8  799.41
#Mann=3,-1,0
  4265.2     0.1       0  4977.8    0.05       0  5022.3     0.1       0
#XS Ineff=2,0
    0.00 4912.30  778.30 5087.80    0.00  778.84
Bank Sta=4977.8,5022.3
XS Rating Curve= 0
Exp/Cntr=0.5,0.3
